--- MOUNTAINRN.prj (project) ---

Proj Title=MOUNTAINRN
Current Plan=p01
Default Exp/Contr=0,0
English Units
Geom File=g01
Flow File=f01
Plan File=p01
BEGIN DESCRIPTION:
END DESCRIPTION:
DSS Export Rating Curves= 0
DSS Export Rating Curve Sorted= 0
DSS Export Volume Flow Curves= 0
DXF OffsetX= 0
DXF OffsetY= 0
DXF ScaleX= 0
DXF ScaleY= 0

--- MOUNTAINRN.p01 (plan) ---

Plan Title=Floodplain
Program Version=4.00
Geom File=g01
Flow File=f01
K Sum by GR=0
Std Step Tol=0.01
Critical Tol=0.01
Num of Std Step Trials=20
Max Error Tol=0.3
Flow Tol Ratio=0.001
Split Flow NTrial=30
Split Flow Tol=0.02
Split Flow Ratio=0.02
Log Output Level=0
Friction Slope Method=1
Unsteady Friction Slope Method=2
Unsteady Bridges Friction Slope Method=1
Global Log Level=0
CheckData=False
Run HTab=0
Run UNet=0
Run PostProcess=0
UNET Theta=0
UNET Theta Warmup=0
UNET ZTol=0
UNET ZSATol=0
UNET MxIter=0
UNET MaxInSteps=0
UNET DtIC=0
UNET DtMin=0
UNET MaxCRTS=0
UNET WFStab=0
UNET SFStab=0
UNET WFX=0
UNET SFX=0
UNET DSS MLevel=0
UNET DZMax Abort=0
UNET Convert EG Bridges=0
UNET Use Existing IB Tables=0
UNET Froude Limit=0
UNET Froude Power=0
Write IC File=0
Echo Input=False
Echo Output=False
Write Detailed=0

--- MOUNTAINRN.f01 (steady flow) ---

Flow Title=NFF Regression Equation
Program Version=4.00
Number of Profiles=1
Profile Names=P100yr
River Rch & RM=MOUNTAINRN,Main      ,26147.8
514.4392
River Rch & RM=MOUNTAINRN,Main      ,25704.9
537.2139
River Rch & RM=MOUNTAINRN,Main      ,23864.9
585.9144
River Rch & RM=MOUNTAINRN,Main      ,23167.8
669.4061
River Rch & RM=MOUNTAINRN,Main      ,20772.3
725.0361
River Rch & RM=MOUNTAINRN,Main      ,20471.9
835.4880
River Rch & RM=MOUNTAINRN,Main      ,19875.5
901.0056
River Rch & RM=MOUNTAINRN,Main      ,17312.9
954.7054
River Rch & RM=MOUNTAINRN,Main      ,17037.5
1066.490
River Rch & RM=MOUNTAINRN,Main      ,12674.6
1166.564
River Rch & RM=MOUNTAINRN,Main      ,12206.1
1297.345
River Rch & RM=MOUNTAINRN,Main      ,9107.8
1398.739
River Rch & RM=MOUNTAINRN,Main      ,8065.9
1543.329
River Rch & RM=MOUNTAINRN,Main      ,5770.7
1667.651
River Rch & RM=MOUNTAINRN,Main      ,552.7
1832.853
River Rch & RM=MOUNTAINRN,Main      ,142.2
1834.591
Boundary for River Rch & Prof#=MOUNTAINRN,Main      ,1
Up Type=0
Dn Type=3
Dn Slope=0.008811

--- MOUNTAINRN.g01 (geometry) ---

Geom Title=USGS 10m DEM
Program Version=4.10

River Reach=MOUNTAINRN      ,Main
Reach XY= 30
     2337382.605      381287.683     2337540.591      381747.752
     2337757.605      381834.557      2338054.48      382890.113
     2338342.675      382938.724     2338356.563      383622.752
     2338788.855      383867.544     2339077.049      385004.696
     2339731.564      385391.849     2339858.299      386279.002
     2340064.897       386369.28     2340174.272      387219.974
     2340518.022      387919.627     2340195.105       388627.96
     2340823.577      388933.516     2340936.425      389442.196
     2340912.119      390089.766     2340667.327      390364.071
     2341858.299      390933.516     2342012.814      391176.571
     2343360.036      394773.793     2343226.355      395897.058
     2343663.855       395971.71     2343761.077      397164.419
     2344405.175      397317.196     2343518.022      398718.238
     2344092.675      399140.113     2344250.661      399740.807
     2343486.772       399846.71     2343224.619      400064.078

Type RM Length L Ch R = 1 ,26147.8 ,446.8,442.9,423.8
XS GIS Cut Line= 3
     2337170.204       381348.78     2337235.016      381380.618
     2337689.302      381197.738
#Sta/Elev= 30
       0  844.88    41.8  840.33    72.2  835.35    96.1  833.66   104.1  832.36
   147.9   820.7   179.7  807.64   191.6  803.68   203.6   801.3   211.6  800.47
  226.72800.8185   235.4   800.9     240  799.89   247.4   797.9   255.4  797.17
   259.3  797.67   263.3  799.92   267.3  801.47   287.2  801.13   303.1  801.75
   319.1  800.76   350.9   804.1   362.8  806.96   390.7  816.56  409.19822.0422
   438.5  830.14   454.4   833.3   510.2  842.68  556.67848.6844   561.9  849.57
#Mann= 6 ,-1 , 0
       0     .12       0  226.72     .07       0     240    .045       0
   263.3     .12       0  409.19     .06       0  556.67     .12       0
#XS Ineff= 2 , 0
                          304.24          804.62
Permanent Ineff=
       F       F
Bank Sta=240,263.3
XS Rating Curve= 0 ,0
Exp/Cntr=0.3,0.1

Type RM Length L Ch R = 1 ,25704.9 ,395.1,397.3,399.3
XS GIS Cut Line= 3
      2337288.26      381746.349     2337317.774      381685.585
     2337796.941      381428.641
#Sta/Elev= 30
       0  850.48   89.25  836.85   103.5  834.52   127.5  829.28   175.5  815.27
   195.5  810.28  205.58806.4656   215.5  802.28   222.4  797.72   227.5  794.71
   231.5  793.94   235.5  794.13   243.5  796.92   279.4  798.56   291.4  797.67
   299.4  798.86   315.4  797.65  329.96 798.542  362.85798.9165   375.4  799.14
   387.4  800.41   395.4  802.13   415.4  809.84   435.4  819.11  454.33825.6983
   471.3  829.88   491.3  833.55  535.14839.6324   579.3  846.91   611.3  850.68
#Mann= 9 ,-1 , 0
       0     .06       0   89.25     .12       0  205.58     .08       0
   222.4    .045       0   243.5     .08       0  329.96     .12       0
  362.85     .06       0  454.33     .12       0  535.14     .06       0
Bank Sta=222.4,243.5
XS Rating Curve= 0 ,0
Exp/Cntr=0.3,0.1

Type RM Length L Ch R = 1 ,25307.6 ,413.1,414.7,416.3
XS GIS Cut Line= 3
     2337449.718      381959.891     2337798.677      381796.696
     2337875.066      381680.377
#Sta/Elev= 30
       0  842.04    35.7  835.21    71.5  829.96    87.4  826.71    99.3   825.1
   111.2  821.62   131.1  817.24   150.9  811.73   158.9   808.5   170.8  805.04
   182.7  799.73   190.6  797.44   214.5  795.62   250.2   794.3   305.8  795.12
   309.8  794.91   317.7   793.4   329.6  790.72   333.6  791.04   337.6  792.19
  339.67  793.83   345.5   798.8   349.5  800.61   369.4  806.92   385.2  810.83
   432.9   824.8  454.84829.3213   480.7  832.39   504.5   836.8   524.4  839.83
#Mann= 4 ,-1 , 0
       0     .12       0   317.7    .045       0  339.67     .12       0
  454.84     .06       0
Bank Sta=317.7,339.67
XS Rating Curve= 0 ,0
Exp/Cntr=0.3,0.1

Type RM Length L Ch R = 1 ,24892.9 ,186.8,187.6,188.3
XS GIS Cut Line= 3
     2337533.052      382246.349     2337974.024      382097.044
     2338107.704      382006.766
#Sta/Elev= 30
       0  839.06    59.7  830.61   107.4  824.87   135.3  819.79   155.2  814.25
   175.1   807.1     183  803.73     195   800.4   206.9  795.68   214.9  793.62
   234.8  791.77   290.5  791.76   314.4  789.85   326.3  787.42   330.3  787.08
   334.2  787.24   338.2  788.14   342.8  789.98   350.2  793.42   362.1  798.05
   397.9  816.35   421.8  825.78   429.8  828.42   441.7  831.51   465.6  836.48
   481.3  838.78   493.1     839   552.1  843.87   583.6   847.4   626.9  853.14
#Mann= 3 ,-1 , 0
       0     .12       0   314.4    .045       0   342.8     .12       0
#XS Ineff= 2 , 0
          279.46  796.33
Permanent Ineff=
       F       F
Bank Sta=314.4,342.8
XS Rating Curve= 0 ,0
Exp/Cntr=0.3,0.1

Type RM Length L Ch R = 1 ,24705.3 ,335.1,334.4,335.8
XS GIS Cut Line= 3
     2337684.755      382384.411     2338030.448      382278.467
     2338160.656      382233.328
#Sta/Elev= 30
       0  825.47    19.9   822.5    31.8  821.28    43.7  818.39    63.6  812.42
    67.5  811.49    75.5  810.64   103.3  801.23   135.1  792.08     143  791.06
   166.9  789.85   206.6  789.67   210.6  789.47   216.8  788.24   230.4  785.96
   234.4  786.03   238.4  786.91   242.4  788.95   246.3  791.93   254.3  795.86
   266.2  802.67   282.1  810.37   305.9  820.56   313.9  824.63   321.8  827.62
   349.6  835.68   377.3  840.34   400.9  840.65   436.4  842.93   499.4  844.45
#Mann= 3 ,-1 , 0
       0     .12       0   216.8    .045       0   242.4     .12       0
Bank Sta=216.8,242.4
XS Rating Curve= 0 ,0
Exp/Cntr=0.3,0.1

Type RM Length L Ch R = 1 ,24370.9 ,249.6,252.3,253
XS GIS Cut Line= 3
     2337763.954      382696.002     2338140.691      382574.474
     2338201.454      382534.544
#Sta/Elev= 30
       0  832.14      20  829.29      36  826.63      64  820.89      76   819.1
      88   816.4     112  809.04     132  801.31     144  796.02   151.9  792.96
   155.9  791.53   159.9  790.61   167.9   789.5   179.9  788.42   187.9  787.99
   199.9  788.09   203.9  787.49   210.6  785.14   215.9  783.65   219.9  783.11
   235.9  785.41   243.9  786.33   255.9   786.4   275.9  789.62   307.9  799.42
   347.9  809.99   359.9  812.91   399.7   821.1   426.5  825.07   468.6   829.9
#Mann= 3 ,-1 , 0
       0     .12       0   210.6    .045       0   235.9     .12       0
Bank Sta=210.6,235.9
XS Rating Curve= 0 ,0
Exp/Cntr=0.3,0.1

Type RM Length L Ch R = 1 ,24118.6 ,269.4,253.7,236.1
XS GIS Cut Line= 4
     2337843.816      382807.113     2337977.496      382859.196
     2338074.078      382832.328     2338209.495      382695.609
#Sta/Elev= 30
       0  823.44    23.9  820.51    55.8  814.83    75.7   809.6   107.6  800.51
   127.5  793.64   143.5  789.54   158.9  787.57   170.5   787.4   178.2  786.82
   189.7  783.75   205.2  781.77     209  781.78   215.4  783.77   224.4  786.67
   232.2  787.38   247.6  787.08   263.4  786.06   279.1  786.47   306.6  786.18
   314.4  786.58   326.2   785.2     338  784.82   353.7  787.32   365.5  790.09
     389  793.25   396.9  794.82   412.6   799.9   428.3  805.85   436.2  807.73
#Mann= 3 ,-1 , 0
       0     .12       0   189.7    .045       0   215.4     .12       0
#XS Ineff= 2 , 0
                          232.99          789.57
Permanent Ineff=
       F       F
Bank Sta=189.7,215.4
XS Rating Curve= 0 ,0
Exp/Cntr=0.3,0.1

Type RM Length L Ch R = 1 ,23864.9 ,238.2,282.7,327.7
XS GIS Cut Line= 3
     2338130.068       383045.87     2338343.759      382755.958
     2338394.391      382741.182
#Sta/Elev= 30
       0  816.68    27.7  812.04   51.17806.3831    71.2  801.24   81.71799.2978
      91  796.01    98.9  791.32   102.9  790.18  127.32 789.911   130.6  789.87
   138.5     786   146.4   783.7   178.1  782.52     186   781.2   197.9  779.07
   201.8  778.94   205.8  779.38   209.8     782   213.7  783.02   241.4   782.3
   245.4  782.61   257.2  786.14   261.2  786.71   273.1  786.34     281  786.76
   288.9  789.28   304.8   799.2   332.4  808.79   382.8  821.92   412.9  828.64
#Mann= 6 ,-1 , 0
       0     .06       0   51.17     .12       0   81.71    .016       0
  127.32     .12       0     186    .045       0   209.8     .12       0
#XS Ineff= 2 , 0
                          224.65          785.15
Permanent Ineff=
       F       F
Bank Sta=186,209.8
XS Rating Curve= 0 ,0
Exp/Cntr=0.3,0.1

Type RM Length L Ch R = 1 ,23582.1 ,120.8,112,102.6
XS GIS Cut Line= 4
     2338184.755       383058.89     2338253.612      383050.117
     2338394.391      383174.776     2338485.537      383250.297
#Sta/Elev= 30
       0  811.69    15.4   808.9    30.8  804.84      54  796.16   63.59791.1324
    69.4  787.41      89  780.86   116.4  779.42     136  780.02  145.87778.7435
  149.42   777.4   163.4  774.82   170.9  777.38   175.2   778.6   190.9  779.09
   202.6  781.46   222.2  780.93   237.9  779.64   273.2  779.23   277.2  779.62
   285.1  782.76     289  783.04     293  782.96   300.8  781.48   312.7  781.62
   316.6  782.43   324.5  785.86   336.4  787.43   367.9  795.71   375.8  796.76
#Mann= 5 ,-1 , 0
       0     .12       0   63.59    .016       0  145.87     .12       0
  149.42    .045       0   170.9     .12       0
Bank Sta=149.42,170.9
XS Rating Curve= 0 ,0
Exp/Cntr=0.3,0.1

Type RM Length L Ch R = 1 ,23470.1 ,325.1,302.3,279.9
XS GIS Cut Line= 4
     2338153.505      383198.213     2338271.995      383206.026
     2338330.589      383230.765     2338466.005      383354.463
#Sta/Elev= 30
       0  824.46   11.28821.9809    27.7   819.1    31.7  817.77    39.6  814.42
    47.5  812.06    63.3  805.15      99  787.66   106.9  784.12   114.8  781.39
   118.8  780.37   130.7  778.74   138.6  774.91   142.6  773.87   146.6   773.6
   158.5  774.48   162.1  775.15   170.4  776.22   178.4  778.44  185.06779.3287
   202.3  780.28   222.2  782.02   250.1   785.1  295.92790.8032     306  792.05
   329.9  793.89   345.8   795.4   353.8  795.93   361.8  795.95   365.8  796.31
#Mann= 6 ,-1 , 0
       0     .06       0   11.28     .12       0   138.6    .045       0
   162.1     .12       0  185.06    .016       0  295.92     .12       0
Bank Sta=138.6,162.1
XS Rating Curve= 0 ,0
Exp/Cntr=0.3,0.1

Type RM Length L Ch R = 1 ,23167.8 ,320.1,308.5,297.4
XS GIS Cut Line= 2
     2338204.927      383565.794     2338644.163      383341.835
#Sta/Elev= 30
       0  819.37    23.9  812.87    35.8  808.42    47.7  803.41    75.6   788.8
   104.6  772.46   107.4  771.41   111.3  770.57   119.3  770.92   123.3  771.64
   127.2  773.11   131.2  775.05   135.2   776.2   155.1  776.21   178.9  775.22
   186.9  775.79   218.7  775.48   222.7  775.92   250.5  782.86   270.4  786.78
   290.3   792.1   306.2  792.63     326  795.11     342  797.62   389.7  806.97
   417.5  811.07   441.4  813.77   457.2  816.83   481.1  818.05     493  819.45
#Mann= 3 ,-1 , 0
       0     .12       0   104.6    .045       0   127.2     .12       0
Bank Sta=104.6,127.2
XS Rating Curve= 0 ,0
Exp/Cntr=0.3,0.1

Type RM Length L Ch R = 1 ,22859.3 ,354.8,372.8,389.7
XS GIS Cut Line= 3
     2338344.684      383830.695     2338432.357      383803.641
     2338692.991      383459.602
#Sta/Elev= 30
       0  830.26      12  827.63    31.9  822.25    91.8  808.73   115.7  802.08
   143.7  792.49   179.7  776.56   191.7  772.19   199.7  770.88   227.6   769.3
   247.6  767.85   251.6  768.08   255.6   769.5   258.5  770.86   263.6  772.13
   275.6  770.24   279.6  770.22   295.6  773.65   311.6  773.59   319.6  774.36
   347.5  782.66   359.5  785.03  397.39788.4617   439.4   792.5   447.4  794.24
  455.23794.3366   475.4  796.61   491.4  797.31   503.4  799.75   523.4  802.44
#Mann= 5 ,-1 , 0
       0     .12       0   227.6    .045       0   258.5     .12       0
  397.39     .06       0  455.23     .12       0
#XS Ineff= 2 , 0
                          262.64          774.18
Permanent Ineff=
       F       F
Bank Sta=227.6,255.6
XS Rating Curve= 0 ,0
Exp/Cntr=0.3,0.1

Type RM Length L Ch R = 1 ,22486.5 ,216.4,217.2,217.9
XS GIS Cut Line= 3
     2338546.852      383997.436     2338572.313      383949.056
     2338976.466      383849.619
#Sta/Elev= 30
       0  784.48     7.8  781.67    15.6  777.67    19.5  776.73    66.6  772.53
    74.5  773.38    82.4  773.27   106.2  770.86   122.1  770.04   157.7  770.43
   177.6  770.03   201.3  768.66   229.1  768.48   252.9  766.54   256.8  766.71
   264.8  768.54   268.7   768.5   272.7  767.99   276.6  766.55   280.6  764.65
   284.6   763.9   292.5  764.84   296.6  766.47   312.3  777.82   340.1  790.77
   363.8  802.98   383.7  811.66   399.5  816.16   443.1  827.25   470.9  830.15
#Mann= 3 ,-1 , 0
       0     .12       0   276.6    .045       0   296.6     .12       0
#XS Ineff= 2 , 0
           216.3  770.92
Permanent Ineff=
       F       F
Bank Sta=276.6,296.6
XS Rating Curve= 0 ,0
Exp/Cntr=0.3,0.1

Type RM Length L Ch R = 1 ,22269.3 ,305.9,302.1,298.2
XS GIS Cut Line= 2
     2338582.314      384147.536     2339021.767       384056.39
#Sta/Elev= 30
       0  810.54    15.9   807.4    23.8  805.11    35.8  800.94    63.6   789.8
    87.4  778.37    99.3  773.15   111.2  769.94   119.2  768.38     135  766.46
     147  766.23   198.6     767   202.6  766.29   205.2   764.8   206.5  764.06
   210.5  762.96   214.5  763.14   225.2     765   234.3  766.55   254.2  765.71
   262.1  767.13     282  774.42   317.7  791.84   333.6  798.72   361.4  808.53
   373.3  811.78   389.2  815.41   405.1  818.17     429  821.53   448.8  823.59
#Mann= 3 ,-1 , 0
       0     .12       0   205.2    .045       0   225.2     .12       0
Bank Sta=205.2,225.2
XS Rating Curve= 0 ,0
Exp/Cntr=0.3,0.1

Type RM Length L Ch R = 1 ,21967.3 ,345.1,345.7,361.2
XS GIS Cut Line= 2
     2338623.546      384453.525     2339083.616      384309.211
#Sta/Elev= 30
       0  820.04    15.9  816.42    47.8  807.17    59.8  804.11    67.7  801.52
   115.6  782.11   139.5  771.68   147.4  769.15   167.4  765.61   179.3  764.53
   195.3  764.28   215.2  764.84   231.1  764.65   247.1     765   250.7   764.4
     255  762.33     259  761.03     263  760.96   278.9  762.72   302.8  764.37
   306.8     766   318.8  772.85   334.7   780.8   358.6  791.27   378.6  799.12
   398.5  805.36   414.4  809.16   438.3   812.5   470.2  815.02   482.2  814.96
#Mann= 3 ,-1 , 0
       0     .12       0   250.7    .045       0   278.9     .12       0
Bank Sta=250.7,278.9
XS Rating Curve= 0 ,0
Exp/Cntr=0.3,0.1

Type RM Length L Ch R = 1 ,21621.6 ,297.6,294.4,274.6
XS GIS Cut Line= 3
     2338674.545      384686.815     2338748.329      384694.411
     2339164.996      384540.331
#Sta/Elev= 30
       0  824.66    15.6  822.41    42.9  817.37    62.5  812.95      94  804.87
   137.6  789.43   169.4  776.46   185.2  770.61   193.2  766.93   201.1  761.04
   205.1  758.53     209  757.75   226.1  759.77   240.8  760.26   252.7  759.46
   260.6  760.95   284.4  761.79   304.2  761.93     328  760.94     336  763.83
   355.8  775.12   375.6   784.5   403.4  794.98   415.3   798.8   427.2  801.19
     443  802.53   474.8  802.82   498.6  801.53   510.5   800.1   518.4  798.48
#Mann= 3 ,-1 , 0
       0     .12       0   201.1    .045       0   226.1     .12       0
Bank Sta=201.1,226.1
XS Rating Curve= 0 ,0
Exp/Cntr=0.3,0.1

Type RM Length L Ch R = 1 ,21327.2 ,265.8,261,255.4
XS GIS Cut Line= 3
     2338809.093      385029.697     2338921.626       384869.61
     2339260.482      384705.261
#Sta/Elev= 30
       0  809.22    67.9  798.02    87.9  795.37   111.8  791.44   147.8   783.3
   191.7  771.21   231.4  764.01     271  760.04   298.8  758.81   314.6  756.12
   326.5  754.19   330.5  754.35   334.4  755.37  337.36  756.81   342.4  759.42
   346.3  759.92   350.3  760.08   358.2  759.35   374.1  760.86   397.9  772.48
   413.7  780.96   429.6  788.12   441.5  792.04   465.2  797.06   485.1  798.18
   500.9  798.33   512.8  797.66   524.7  796.27   536.6  793.58   572.3  779.86
#Mann= 3 ,-1 , 0
       0     .12       0   314.6    .045       0  337.36     .12       0
Bank Sta=314.6,337.36
XS Rating Curve= 0 ,0
Exp/Cntr=0.3,0.1

Type RM Length L Ch R = 1 ,21066.2 ,315,293.9,272.4
XS GIS Cut Line= 3
     2338918.116      385132.228     2339019.067      385112.302
     2339292.519      384902.209
#Sta/Elev= 30
       0  805.96    23.8  802.26    35.6   799.9    98.9  781.66   118.8   776.9
   130.6  772.87   150.5  764.67   162.4  760.79   174.2   758.6   194.1   758.1
     198  757.09  204.75  753.44     206  752.75   213.9  752.21   225.8  752.79
   229.8   753.8   237.7  757.44   241.6  758.15   277.3  756.03   285.2  756.48
   297.1  758.64   316.9  764.95   328.8   770.8   352.6  780.23   372.4  784.99
   384.3  787.01   396.2  787.98   427.9  787.64   439.8  785.89   447.7  784.05
#Mann= 3 ,-1 , 0
       0     .12       0  204.75    .045       0   229.8     .12       0
#XS Ineff= 2 , 0
                          242.62          761.79
Permanent Ineff=
       F       F
Bank Sta=204.75,229.8
XS Rating Curve= 0 ,0
Exp/Cntr=0.3,0.1

Type RM Length L Ch R = 1 ,20772.3 ,293.5,300.4,307.4
XS GIS Cut Line= 3
     2339330.578      385417.935     2339316.255      385321.581
      2339338.39      385052.049
#Sta/Elev= 30
       0  799.76    19.5  796.94    42.9  792.88    50.6  791.12    58.4  789.68
    77.9  785.51   121.3  774.54   133.2  770.55   149.1  764.44   153.1  762.45
     161  756.94     165  755.32     177  751.51   180.9  750.37   184.9   749.8
   188.9   749.8   192.9  750.23     199  751.42   212.8  754.25   216.7  754.67
   248.5  754.77   268.4  754.37   300.2  754.89   312.2  755.28   332.1  756.38
     340  757.09     344  757.71   359.9  758.52   363.9  758.84   367.8   759.6
#Mann= 3 ,-1 , 0
       0     .12       0     177    .045       0     199     .12       0
#XS Ineff= 2 , 0
                          223.88          756.99
Permanent Ineff=
       F       F
Bank Sta=177,199
XS Rating Curve= 0 ,0
Exp/Cntr=0.3,0.1

Type RM Length L Ch R = 1 ,20471.9 ,267.4,290.2,313.1
XS GIS Cut Line= 3
     2339476.411      385455.695     2339544.119       385408.82
     2339680.838      385079.393
#Sta/Elev= 30
       0  779.83    23.5  773.93    47.1  768.95    66.7  763.56    86.3   756.8
    94.2  754.96   102.2  753.77     118  752.38   141.8  752.53   173.5  751.32
   177.5  750.27   181.4  748.56   185.4  747.75   201.2  750.46   213.1  750.53
     225  751.51   244.8  750.81   251.6  749.27   256.7  748.11   264.6  747.68
   268.6   748.3   271.6   749.7   276.5  751.74   284.5  752.77   304.3  752.54
   320.1  753.02   328.1  754.23   347.9  758.71   391.5  773.05     439  781.52
#Mann= 3 ,-1 , 0
       0     .12       0   251.6    .045       0   271.6     .12       0
Bank Sta=251.6,271.6
XS Rating Curve= 0 ,0
Exp/Cntr=0.3,0.1

Type RM Length L Ch R = 1 ,20181.6 ,303.7,306.1,308.6
XS GIS Cut Line= 4
     2339524.588      385570.279      2339650.89      385509.081
     2339890.474      385441.372     2340012.869      385489.549
#Sta/Elev= 30
       0  780.49    15.6   777.9    27.3  775.19    58.5  766.91    81.9  758.83
    89.7  756.62   113.1  751.66     168  747.99   175.9  748.85   207.5  749.49
   211.5  749.23   215.4  748.08   219.4  745.43   223.3   743.7   227.3  743.25
   235.2  743.69   242.2  744.97     251  746.41   266.8  746.72   270.8  747.35
   278.7  749.82   290.5   755.3   298.4  758.16   322.1  764.85   361.6  773.76
   389.3     779   397.3  781.36   457.1   795.8   504.9  806.77   520.8  809.93
#Mann= 3 ,-1 , 0
       0     .12       0   219.4    .045       0   242.2     .12       0
Bank Sta=219.4,242.2
XS Rating Curve= 0 ,0
Exp/Cntr=0.3,0.1

Type RM Length L Ch R = 1 ,19875.5 ,392,386.6,381
XS GIS Cut Line= 3
      2339494.64      385824.185     2339933.442       385746.06
     2339975.109      385738.247
#Sta/Elev= 30
       0  800.31    55.7  784.62    75.6  780.91    87.6  779.97   115.4  776.04
   123.4   774.6   139.3  770.34   155.2  764.81     191  750.04   210.9  743.54
   214.9  743.38   226.8  745.54   238.8  745.54   246.7  744.16   250.2  742.33
   254.7  740.27   258.7  739.92   266.6   740.2   274.6  742.64   282.5  744.32
   302.4  743.81   314.4  744.95   338.3  744.68   342.2  745.58   346.2   747.2
   358.2  754.07     386  770.74   401.9  777.06   453.4  792.49   488.1  800.77
#Mann= 3 ,-1 , 0
       0     .12       0   250.2    .045       0   274.6     .12       0
Bank Sta=250.2,274.6
XS Rating Curve= 0 ,0
Exp/Cntr=0.3,0.1

Type RM Length L Ch R = 1 ,19488.9 ,244.2,237.9,231.6
XS GIS Cut Line= 3
     2339615.734      386186.164      2339769.38      386165.331
     2340104.015      386028.612
#Sta/Elev= 30
       0  791.66       4  790.51       8  789.96    23.8  785.34    71.6  770.32
    91.4  765.94   115.3  761.61   151.1  752.09   170.9  744.72  181.86 743.352
   194.8  742.24  208.16740.4722   224.2  739.49   238.5  737.83   246.4  738.42
   250.4  739.85   254.4  741.38   258.3  741.98   282.2  741.47   325.9  744.65
   349.7  747.81   353.7  749.09   369.6   757.3   377.5  760.82   381.5   762.5
   389.4  764.95   417.2  771.29   472.8   785.3   500.6  789.21   516.5  791.93
#Mann= 5 ,-1 , 0
       0     .12       0  181.86     .06       0  208.16     .12       0
   224.2    .045       0   250.4     .12       0
Bank Sta=224.2,250.4
XS Rating Curve= 0 ,0
Exp/Cntr=0.3,0.1

Type RM Length L Ch R = 1 ,19251   ,307.9,318.4,327.5
XS GIS Cut Line= 3
     2339752.453      386428.352     2339855.317      386397.102
     2340160.005      386156.216
#Sta/Elev= 30
       0  791.06    35.8  782.93    51.8  778.53    67.7  773.35   103.5  760.08
   131.3  748.45   147.1   742.5   155.1  741.43   174.9  740.53   187.3  738.26
   198.7  735.88   207.3  737.49   210.6  738.81   214.5  739.52   238.3  738.95
   246.2  739.48   254.2  739.04   301.7  739.37   317.6  740.03   321.5   741.5
   325.5  743.91   337.4  752.92   345.3  757.22   349.3  758.85   388.9   770.4
   404.8  774.82   424.6  779.38   444.4   782.5   472.1  787.82   495.9  791.44
#Mann= 3 ,-1 , 0
       0     .12       0   187.3    .045       0   207.3     .12       0
Bank Sta=187.3,207.3
XS Rating Curve= 0 ,0
Exp/Cntr=0.3,0.1

Type RM Length L Ch R = 1 ,18932.6 ,279.3,280.5,282.5
XS GIS Cut Line= 3
     2339778.494      386506.477     2339949.067      386576.789
     2340299.328      386447.883
#Sta/Elev= 30
       0  781.53    19.6  776.06    35.3  772.71    58.9  765.03   102.1   748.8
   117.8  744.48   141.3  741.61  173.57740.6621  184.74740.5868   196.4  741.15
   200.4  740.46   208.3  737.46  223.34737.2243  288.99736.9574   299.6  737.04
   311.6  740.21  317.13740.0156   331.4  738.47     350  734.61   359.2  732.04
   363.2  731.86   367.1  732.86     370  734.49     383   742.9   394.9  748.26
   414.8  754.35   430.7  757.91   498.2  777.33  523.02781.6658   557.7  787.37
#Mann= 9 ,-1 , 0
       0     .12       0  173.57     .06       0  184.74     .12       0
  223.34     .04       0  288.99     .06       0  317.13     .12       0
     350    .045       0     370     .12       0  523.02     .06       0
#XS Ineff= 2 , 0
          313.48  741.33
Permanent Ineff=
       F       F
Bank Sta=350,370
XS Rating Curve= 0 ,0
Exp/Cntr=0.3,0.1

Type RM Length L Ch R = 1 ,18652   ,249.4,251.7,248.9
XS GIS Cut Line= 2
     2339950.369      386843.716     2340396.984      386731.737
#Sta/Elev= 30
       0  770.12    35.7  761.56    47.6  759.48    59.5  756.62    83.4  750.07
    95.3  747.37     123  736.14     127  735.21  148.64734.6765   170.7  733.76
   194.5  733.85  208.67733.1441   227.1  731.88   234.2   729.8   238.2  729.62
   242.1  731.11   246.1  733.67   247.1  733.92     258  735.61     262  737.01
   281.8  745.66   293.7  751.36   301.7  754.62   317.5  762.28   333.4  766.75
   353.3  773.29     385  780.93   412.8   784.7  439.35787.5475   460.4  788.37
#Mann= 6 ,-1 , 0
       0     .12       0  148.64     .06       0  208.67     .12       0
   227.1    .045       0   247.1     .12       0  439.35     .06       0
Bank Sta=227.1,247.1
XS Rating Curve= 0 ,0
Exp/Cntr=0.3,0.1

Type RM Length L Ch R = 1 ,18400.3 ,339.7,328.6,318
XS GIS Cut Line= 3
     2339977.713      387049.445     2340372.244       386971.32
     2340486.828      387023.404
#Sta/Elev= 30
       0  778.56    15.9  773.76    39.8  768.24    83.6  755.75   123.4  746.53
   135.4  744.26   147.3  739.26   151.3  736.66   159.3  730.24   161.7  729.24
   167.2   727.9   171.2  727.77   183.2  728.88   191.1   730.8   199.1  731.85
     227  732.33   238.9  733.63   274.8  734.32   314.6   737.2   322.6  739.03
   334.5   742.8   354.4  747.14  395.01753.0434   402.2  754.09   429.7  760.84
   441.5  764.36  468.69 767.159   484.8  769.33   496.6   774.1   528.1  779.09
#Mann= 5 ,-1 , 0
       0     .12       0   161.7    .045       0   183.2     .12       0
  395.01    .016       0  468.69     .12       0
Bank Sta=161.7,183.2
XS Rating Curve= 0 ,0
Exp/Cntr=0.3,0.1

Type RM Length L Ch R = 1 ,18071.8 ,276,282.8,289.9
XS GIS Cut Line= 4
     2340038.911      387359.341     2340208.182      387295.539
     2340339.692      387204.393     2340484.224      387154.914
#Sta/Elev= 30
       0   781.4     7.9  778.49    27.5  773.04      59  762.36    90.4  754.72
   141.6  746.23   149.4  744.29   161.2   740.6   180.9  732.27   200.4  730.11
   208.2   730.5   235.5     730     255  728.41   262.8  726.84   270.7  725.37
   274.6  725.33   282.8  726.32   290.2  730.91   294.1   731.9   313.6  733.22
   333.1   738.8  347.23744.4092   356.6  747.74   372.2  749.15   376.2  751.05
  379.99754.3541     384  756.65  410.72766.7629  449.76774.7928   493.7  781.76
#Mann= 7 ,-1 , 0
       0     .12       0   262.8    .045       0   282.8     .12       0
  347.23    .016       0  379.99     .12       0  410.72     .06       0
  449.76     .12       0
Bank Sta=262.8,282.8
XS Rating Curve= 0 ,0
Exp/Cntr=0.3,0.1

Type RM Length L Ch R = 1 ,17789   ,317,317,316.3
XS GIS Cut Line= 3
     2340021.984      387477.831     2340114.432      387505.174
     2340506.359       387377.57
#Sta/Elev= 30
       0  788.96    42.4  779.85    77.1  770.13    88.7   767.3     140  756.74
   175.7  748.36   191.5   746.2   199.4  744.65   203.4   743.2   223.2  732.98
   227.2  731.34   235.1  729.34   243.6  725.46     247  724.56   258.9  724.18
   266.8  724.64   270.8  725.92   278.7  727.13   302.5  725.99   318.4  727.77
   346.1  727.23     358  727.49   366.3 730.116   377.8  731.92   393.6  732.11
  401.82 734.039   433.3  746.47     469   759.2   496.7  769.67   508.6  771.57
#Mann= 5 ,-1 , 0
       0     .12       0   243.6    .045       0   270.8     .12       0
   366.3    .016       0  401.82     .12       0
Bank Sta=243.6,270.8
XS Rating Curve= 0 ,0
Exp/Cntr=0.3,0.1

Type RM Length L Ch R = 1 ,17472   ,170.4,159.1,147.5
XS GIS Cut Line= 3
     2340072.765      387845.018     2340214.692      387742.154
     2340576.671      387626.268
#Sta/Elev= 30
       0  749.42    23.9  738.63    27.9  737.49   43.02736.7266   64.51734.4114
    99.6   733.1   107.6  731.39   119.5  736.11   171.3  746.33   187.2  747.38
   218.8  747.72   230.7  747.21   254.5   743.3   266.3   739.1   282.2  731.02
   294.1  726.17  317.99725.1143  348.36   724.7   373.2  724.46   381.2  723.39
     397  722.13     401  722.68  402.82  723.75  404.83 724.762   408.9  727.41
   424.7     727  440.73734.6563   476.2  748.73   503.9  758.56   555.4  771.32
#Mann= 9 ,-1 , 0
       0     .12       0   43.02     .06       0   64.51     .12       0
  317.99     .06       0  348.36     .12       0   381.2    .045       0
  402.82     .12       0  404.83    .016       0  440.73     .12       0
Bank Sta=381.2,402.82
XS Rating Curve= 0 ,0
Exp/Cntr=0.3,0.1

Type RM Length L Ch R = 1 ,17312.9 ,125.3,143.1,160.9
XS GIS Cut Line= 3
     2340140.484      387901.686     2340373.557      387882.154
     2340577.984      387689.446
#Sta/Elev= 30
       0  740.61    11.9  734.92    15.9  733.74    27.8  733.15    39.6  731.04
   54.56729.7729    83.2  727.08    91.2  728.71     111  729.78   118.9  732.24
   130.8  737.92   142.7   741.2   162.5  743.98   178.4  744.37   202.2  741.68
   233.9  729.84   253.7   725.5   265.5  723.88   289.3  723.01   297.2  723.49
   302.1  722.64   309.1  720.79     317   721.6   322.1  723.17   324.9  724.21
  333.09724.4211   372.4  723.79  393.34728.3791   423.8  738.75   514.8  762.99
#Mann= 6 ,-1 , 0
       0     .06       0   54.56     .12       0   302.1    .045       0
   322.1     .12       0  333.09    .016       0  393.34     .12       0
Bank Sta=302.1,322.1
XS Rating Curve= 0 ,0
Exp/Cntr=0.3,0.1

Type RM Length L Ch R = 1 ,17169.9 ,117.8,132.4,147
XS GIS Cut Line= 3
     2340146.995      387940.748      2340606.63      387926.425
     2340719.912      388027.988
#Sta/Elev= 30
       0  742.86    4.23741.6293      16  738.18      28  733.17   65.45728.4678
      80  725.42      92  727.47     124  727.35     136  729.12     160  736.21
   179.9  737.86   199.9  735.36   227.9  726.28  236.52724.6616   255.9  722.99
  292.54723.3052  324.81723.0656   335.9  723.65     357  720.62   371.9  719.16
   382.8  720.91   391.9  722.79   407.9  722.74   443.9  726.91   463.8  728.26
   479.4  733.26   498.9  736.67   545.7   747.9   588.6  756.23     612   759.2
#Mann= 8 ,-1 , 0
       0     .12       0    4.23     .06       0   65.45     .12       0
  236.52     .06       0  292.54    .016       0  324.81     .12       0
     357    .045       0   382.8     .12       0
#XS Ineff= 2 , 0
          281.26  724.86
Permanent Ineff=
       F       F
Bank Sta=357,382.8
XS Rating Curve= 0 ,0
Exp/Cntr=0.3,0.1

Type RM Length L Ch R = 1 ,17037.5 ,168.7,164.9,161.1
XS GIS Cut Line= 3
     2340156.109      387996.738     2340339.703      387977.206
     2340663.922      388163.404
#Sta/Elev= 30
       0  742.81    39.3  732.33      55  731.24    82.5  723.66   102.1  725.82
   125.7  725.54   149.3  726.24   168.9  729.05   180.7  729.88   184.6  729.68
   204.5  724.64  232.91  723.24  269.48722.4134     304  720.85   311.9   721.2
  321.74720.0508   325.3  719.26   331.8  716.88   335.8  716.27   339.8  716.35
   347.7  719.14   351.7  721.48   367.6  734.72   375.6  739.32   391.5  746.02
   423.3  755.23   443.2  758.93     467  761.54  520.21762.8967   558.5  764.58
#Mann= 7 ,-1 , 0
       0     .12       0  232.91     .06       0  269.48    .016       0
  321.74     .12       0   325.3    .045       0   347.7     .12       0
  520.21     .06       0
Bank Sta=325.3,347.7
XS Rating Curve= 0 ,0
Exp/Cntr=0.3,0.1

Type RM Length L Ch R = 1 ,16872.6 ,333.9,325.5,316.8
XS GIS Cut Line= 3
     2340143.078      388092.414     2340510.265      388239.549
     2340643.078      388231.737
#Sta/Elev= 30
       0  740.81   29.07735.9188      40   734.3    63.9  732.51   80.87730.0372
   107.9  724.95   139.8  722.77   167.8  719.32  187.36720.0002   195.8  720.37
   211.8  719.43   227.8  720.34   231.8  719.21  235.66 717.181   235.9  717.09
   239.7  715.67   243.7  715.48   255.7  716.17   259.7  717.05   267.7  719.17
   283.7  721.98   295.7  726.88   319.6  739.69   351.6   751.8   367.6  756.78
   387.6  759.55   426.9  762.39   462.1   762.8  485.78761.7549   528.6  762.12
#Mann= 8 ,-1 , 0
       0     .12       0   29.07     .08       0   80.87     .12       0
  187.36    .016       0  235.66     .12       0   235.9    .045       0
   259.7     .12       0  485.78     .06       0
#XS Ineff= 2 , 0
          191.01  722.32
Permanent Ineff=
       F       F
Bank Sta=235.9,259.7
XS Rating Curve= 0 ,0
Exp/Cntr=0.3,0.1

Type RM Length L Ch R = 1 ,16547.1 ,413.5,391,368
XS GIS Cut Line= 4
     2339990.005      388439.467     2340131.793      388471.551
     2340398.056      388481.293     2340549.243      388397.808
#Sta/Elev= 30
       0  773.62    11.8   770.4    31.4  763.55      55  753.52    94.3  734.11
     110  728.47   121.8  725.23   153.3  719.64  188.63717.2036   220.9  717.53
   228.1 718.394   232.9   718.2   242.4   715.2   252.8  713.02   256.7  713.15
   264.7  714.83   272.6  717.11   276.6  717.71   296.5  717.55   312.4  718.73
   364.1  718.13     376  717.32     380  717.63     388  719.26   435.4  733.74
   462.8  739.46   509.9     748   533.5  750.79   545.3  751.55   584.5  752.72
#Mann= 5 ,-1 , 0
       0     .12       0  188.63    .016       0   228.1     .12       0
   242.4    .045       0   264.7     .12       0
#XS Ineff= 2 , 0
                          307.32          723.84
Permanent Ineff=
       F       F
Bank Sta=242.4,264.7
XS Rating Curve= 0 ,0
Exp/Cntr=0.3,0.1

Type RM Length L Ch R = 1 ,16156.2 ,177.2,177.9,178.8
XS GIS Cut Line= 3
     2340223.807      388880.174     2340520.682      388572.883
     2340725.109      388553.352
#Sta/Elev= 30
       0  742.65   10.89741.8138   13.54741.5229    39.9   738.5    51.9  732.83
    55.9   731.8    75.9  729.78  108.98724.7815   115.8  724.21   123.8  722.27
   139.8   722.1  145.86 720.829   151.7  718.56   167.7  715.69   223.6  714.59
   249.9  712.37   267.6  710.64   271.5   711.4  273.17  712.68   279.5  714.92
   323.4  714.34   367.4  716.62   399.3  720.77   427.3  726.86   458.9  737.09
   502.3  749.06     526  754.46   545.8  758.24   597.1  765.84   632.6  769.87
#Mann= 7 ,-1 , 0
       0     .12       0   10.89     .06       0   13.54     .12       0
  108.98    .016       0  145.86     .12       0   249.9    .045       0
  273.17     .12       0
Bank Sta=249.9,273.17
XS Rating Curve= 0 ,0
Exp/Cntr=0.3,0.1

Type RM Length L Ch R = 1 ,15978.3 ,427.5,437.7,446.1
XS GIS Cut Line= 3
     2340347.505      389024.706     2340395.682       388933.56
     2340722.505      388626.268
#Sta/Elev= 30
       0  763.22    31.7  756.56    59.5  748.97   95.07740.6341   103.1  738.82
     119  737.75   130.9  732.24   143.1 729.736   150.7   727.8   158.7  722.46
   178.5  721.74   182.5  721.06  190.07718.0026   210.3  710.34   214.2  709.44
   222.2  709.36   232.2  710.75     246   712.7   269.8   713.7   285.7  711.85
   301.6  713.39   345.3  713.49     373  712.38   392.9   712.9   396.9  714.34
   424.7  729.76   436.6  733.89   480.2  751.73     508  760.38   551.7  768.62
#Mann= 6 ,-1 , 0
       0     .06       0   95.07     .12       0   143.1    .016       0
  190.07     .12       0   210.3    .045       0   232.2     .12       0
Bank Sta=210.3,232.2
XS Rating Curve= 0 ,0
Exp/Cntr=0.3,0.1

Type RM Length L Ch R = 1 ,15540.6 ,83.9,86.1,88.6
XS GIS Cut Line= 3
     2340495.942      389137.987     2340904.796      388949.185
     2340924.328      388852.831
#Sta/Elev= 30
       0  748.97    8.46748.0698    43.8  744.62   90.32 736.126  102.07732.9728
   127.5  725.56   135.5  719.83   139.5  718.97  155.06717.9757   163.4  715.58
   171.4  714.33   219.2  712.82     267  710.47   302.9  709.96  327.94710.4114
   346.7  709.94   350.7  709.24   358.7  706.59   366.6  705.58   381.9  706.93
   394.6  709.63   410.5  711.16   418.5  715.13   422.4  715.96   450.3  719.57
   485.7  729.62   497.5   731.3   517.2  733.11   536.9  736.98   548.7   737.7
#Mann= 8 ,-1 , 0
       0     .12       0    8.46     .06       0   90.32     .12       0
  102.07    .016       0  155.06     .06       0  327.94     .12       0
   358.7    .045       0   381.9     .12       0
Bank Sta=358.7,381.9
XS Rating Curve= 0 ,0
Exp/Cntr=0.3,0.1

Type RM Length L Ch R = 1 ,15454.5 ,106.1,110.6,114.8
XS GIS Cut Line= 3
     2340559.744      389187.466     2340752.453      389101.529
     2341059.744      388988.247
#Sta/Elev= 30
       0  744.16       8  738.99    23.9   735.8    35.8  734.65    75.6  734.94
    87.6  732.09   92.59729.1676   103.5  721.48   107.5  720.24  129.29719.0601
  146.71717.4219  161.38715.7101  193.46712.5453  224.07710.6858  256.44709.2061
   294.9  705.87   298.9  704.66   306.9  703.98   319.7  705.14   338.8  710.34
   362.8  709.19   374.8  710.18   394.7  714.24  421.21712.5763   430.7  713.16
  454.13717.8018   482.6  718.29   502.6  721.51   522.5  726.28   538.5  727.75
#Mann= 12 ,-1 , 0
       0     .06       0   92.59    .016       0  129.29     .06       0
  146.71     .12       0  161.38     .06       0  193.46     .12       0
  224.07     .06       0  256.44     .12       0   298.9    .045       0
   319.7     .12       0  421.21    .016       0  454.13     .12       0
Bank Sta=298.9,319.7
XS Rating Curve= 0 ,0
Exp/Cntr=0.3,0.1

Type RM Length L Ch R = 1 ,15343.9 ,168.2,168.2,168.3
XS GIS Cut Line= 3
     2340593.599      389298.143     2340669.119      389212.206
     2341077.974      389136.685
#Sta/Elev= 30
       0   759.5     7.9  759.14   28.59753.5348    55.2  747.81    67.1  746.67
    87.8  741.08   110.5  736.76  121.66736.4348   134.4  735.76   138.4  734.35
   146.4  728.39   174.4  728.62   184.4 724.415   210.4   715.7   226.3  712.16
   250.3     709   278.3  707.92   294.3  703.75   306.3  702.55   317.6  704.33
   326.3  707.82  381.79708.6667   402.2  714.12  423.82711.8605  453.74712.7464
   462.2  716.18   470.2  717.11   502.2  732.71   514.2  735.56   530.2  743.28
#Mann= 10 ,-1 , 0
       0     .08       0   28.59     .12       0    87.8     .06       0
  121.66    .016       0   184.4     .12       0   294.3    .045       0
   317.6     .12       0  381.79    .016       0  423.82     .04       0
  453.74     .12       0
Bank Sta=294.3,317.6
XS Rating Curve= 0 ,0
Exp/Cntr=0.3,0.1

Type RM Length L Ch R = 1 ,15175.6 ,213.5,214.5,215.4
XS GIS Cut Line= 3
     2340601.411      389425.747     2340729.015       389371.06
     2341137.869      389295.539
#Sta/Elev= 30
       0  767.91    35.7  761.95   87.79750.9482   103.1  748.54  119.68747.2234
     123  746.02   130.9  740.78  150.78738.8437   154.8  737.09   174.8   723.6
   198.8  711.68   210.8  704.77   214.8  704.04   230.8  704.14   242.8  705.78
   262.8  706.22   286.8  704.89  301.72702.9668   307.5  701.89   314.7  701.51
   327.5   701.9   334.7  704.25  344.03705.1266   370.7   705.5   410.7  716.16
   426.7  723.24   470.6  735.43   478.6  738.42   490.6  739.82   554.6  755.26
#Mann= 8 ,-1 , 0
       0     .06       0   87.79     .12       0  119.68    .016       0
  150.78     .12       0  301.72    .016       0   307.5    .045       0
   327.5    .016       0  344.03     .12       0
Bank Sta=307.5,327.5
XS Rating Curve= 0 ,0
Exp/Cntr=0.3,0.1

Type RM Length L Ch R = 1 ,14961.1 ,360.6,362.5,364.3
XS GIS Cut Line= 2
     2340645.682      389587.206     2341143.078      389515.591
#Sta/Elev= 30
       0  759.26   65.96747.0102    83.8  744.15    87.7  743.25    95.7   739.5
   99.51739.5476   115.7  738.08  132.95728.9264   155.5   715.9   171.5  707.66
   187.4     702   199.4  701.51   215.4  704.36   255.2  703.84   259.2  703.76
  269.72  700.58   287.2  700.09   293.7  700.53     323  703.83     339  703.24
     351  706.37   366.9  708.82   378.9     712   398.8  719.41   426.8  732.86
   434.7  735.85   442.7  736.59   454.7  741.16   466.6  743.83   502.5  750.48
#Mann= 6 ,-1 , 0
       0     .06       0   65.96     .12       0   99.51    .016       0
  132.95     .12       0  269.72    .045       0   293.7     .12       0
Bank Sta=269.72,293.7
XS Rating Curve= 0 ,0
Exp/Cntr=0.3,0.1

Type RM Length L Ch R = 1 ,14598.6 ,103.8,104.7,104.7
XS GIS Cut Line= 4
     2340771.995      389863.578     2340818.859       389902.31
     2341143.078      389894.497     2341199.067      389868.456
#Sta/Elev= 30
       0  722.33     3.8  720.21    5.88719.8378    22.8  719.58      38  717.28
    45.6  714.75    60.8  708.21    76.6  704.01    84.5  702.46    92.4  701.62
   100.4  701.71  114.01700.7122     132  700.38   163.6  701.35   186.1  698.64
   195.3  697.12   199.2  697.23   206.1  698.48     223  701.52   234.8  702.39
   250.6  702.23   258.6  703.63   266.5  705.73   278.3  709.78   313.9  724.75
   345.6  734.98   365.3  739.46   385.1  742.58   408.3   748.7   446.9  756.88
#Mann= 5 ,-1 , 0
       0     .12       0    5.88    .016       0  114.01     .12       0
   186.1    .045       0   206.1     .12       0
Bank Sta=186.1,206.1
XS Rating Curve= 0 ,0
Exp/Cntr=0.3,0.1

Type RM Length L Ch R = 1 ,14494   ,244.2,262.6,281.6
XS GIS Cut Line= 3
     2340722.516      389969.047     2340775.901       389996.39
     2341127.464      389984.672
#Sta/Elev= 30
       0  710.26       8  707.96      16  707.55      28  707.76      36  707.54
      44  706.83      52  705.53   55.27705.3992      84  704.43      92  703.84
   111.9  701.62   135.9  700.26   151.9  699.72   171.9  700.34   175.9  699.85
   180.6  697.77   183.9  696.61   191.9  696.16   207.9   696.9   223.9  698.05
   235.9  699.64   271.8  701.39   283.8   703.1   299.8   707.1   319.8   713.2
   335.8   717.2   343.8  718.66   355.8  722.01   383.8  731.59   411.7  739.66
#Mann= 4 ,-1 , 0
       0     .06       0   55.27     .12       0   180.6    .045       0
   207.9     .12       0
Bank Sta=180.6,207.9
XS Rating Curve= 0 ,0
Exp/Cntr=0.3,0.1

Type RM Length L Ch R = 1 ,14231.4 ,153.5,146,138.3
XS GIS Cut Line= 2
     2340632.661      390062.466     2340856.619      390247.362
#Sta/Elev= 30
       0  703.53       4  702.94    23.9  701.47    47.7   700.6    59.7  699.33
    67.6  700.41    75.6  702.21    79.6  702.54    91.5  701.59   107.4  701.19
   163.1  698.68   171.1  698.75     175  698.53     179  697.24     187   693.7
   198.9  692.84   202.9  692.88   206.9  693.38   211.1   694.4   218.8  696.89
   222.8  697.74   234.7  697.73   238.7  698.18   242.7  700.27   246.7  703.26
   250.6  705.49   266.6  712.55   278.5  717.15   282.5  718.37   290.4   719.8
#Mann= 3 ,-1 , 0
       0     .12       0     187    .045       0   211.1     .12       0
Bank Sta=187,211.1
XS Rating Curve= 0 ,0
Exp/Cntr=0.3,0.1

Type RM Length L Ch R = 1 ,14085.4 ,219.6,188.1,156.8
XS GIS Cut Line= 3
     2340540.224      390221.998     2340781.109      390326.165
     2340863.141      390264.967
#Sta/Elev= 30
       0  705.68    35.8  703.08    59.6  702.51    79.5  700.29    99.4  699.03
   143.2  698.08   151.1  696.81   159.1  694.02     163  693.18   178.9  692.63
   182.9  693.19  185.37  694.02   186.9  695.24   190.9  696.84   194.8  697.09
   206.8  697.07   222.7  696.43   238.6  697.81   254.5  697.35   266.4  696.31
   282.1  697.72     290  697.82   301.8  697.38   309.7  698.06   313.6  698.84
   321.5  701.46   329.4  704.64   345.1  711.89   356.9   716.1   364.8  718.47
#Mann= 3 ,-1 , 0
       0     .12       0   159.1    .045       0  185.37     .12       0
Bank Sta=159.1,185.37
XS Rating Curve= 0 ,0
Exp/Cntr=0.3,0.1

Type RM Length L Ch R = 1 ,13897.3 ,373.8,378.9,379.3
XS GIS Cut Line= 3
     2340709.495      390621.738     2340712.099      390464.186
     2340885.276      390276.686
#Sta/Elev= 30
       0   721.6    11.8  716.23    31.5  707.98    43.3  703.55    51.2  701.07
    59.1  699.08    70.9  697.27   89.05695.7457  129.71694.5648   145.8  695.72
   165.6  696.17   181.5  694.24   193.7  691.51   201.4  690.66   217.4  691.68
   221.4  692.45   225.4  694.33   229.4  695.43   249.3  696.71   297.2   696.6
   309.1  695.64   321.1  696.75     345  696.94     357  696.42     361  697.09
   368.9  699.88   372.9  701.65   388.9  710.44   404.8     718   412.8  721.05
#Mann= 5 ,-1 , 0
       0     .12       0   89.05     .04       0  129.71     .12       0
   193.7    .045       0   217.4     .12       0
#XS Ineff= 2 , 0
           161.1  697.28
Permanent Ineff=
       F       F
Bank Sta=193.7,217.4
XS Rating Curve= 0 ,0
Exp/Cntr=0.3,0.1

Type RM Length L Ch R = 1 ,13518.5 ,365.1,368.5,375
XS GIS Cut Line= 3
      2340900.89      390710.904     2340967.296      390680.956
     2341180.849       390404.29
#Sta/Elev= 30
       0  731.71      69  720.03    84.8  716.61   108.6  709.66   128.4  701.08
   140.4  696.67   160.2  694.31   172.1  693.55   176.1  692.17   180.1  689.78
     184  688.89     188  688.67   199.9   689.6   207.9  688.23   211.8  688.26
   223.8  690.32   235.7  691.05   251.6  690.21   263.5  692.58   275.4  692.37
   283.3  693.14   291.3  696.73   319.1  714.23     331     721   338.9  726.81
   346.9  731.82   370.7  744.74   390.6  753.43   410.4  758.09   422.3  760.15
#Mann= 3 ,-1 , 0
       0     .12       0   199.9    .045       0   223.8     .12       0
Bank Sta=199.9,223.8
XS Rating Curve= 0 ,0
Exp/Cntr=0.3,0.1

Type RM Length L Ch R = 1 ,13150   ,227.3,219.9,208.2
XS GIS Cut Line= 4
     2341132.661      390934.862     2341167.817      390867.154
     2341405.083        390611.1     2341419.119      390493.456
#Sta/Elev= 30
       0  729.85    11.4  727.97      61  722.19    80.3  719.34    96.1  716.12
   127.9  707.58   147.7  700.38   167.5  692.15   171.5  690.84   175.5  689.94
   187.4   689.6   191.3  688.19   195.3  686.01   199.3  685.13   211.2  685.07
   219.3  686.22     227  687.84   258.8  688.22   270.7  690.33   290.5  691.17
   330.2   697.6   338.1  699.88   357.9  708.14   381.7  716.99   401.6  722.32
   405.5  723.76   433.3  731.55   492.5   745.1   520.2  750.15   543.8  755.03
#Mann= 3 ,-1 , 0
       0     .12       0   195.3    .045       0   219.3     .12       0
Bank Sta=195.3,219.3
XS Rating Curve= 0 ,0
Exp/Cntr=0.3,0.1

Type RM Length L Ch R = 1 ,12930.1 ,256.8,255.5,255.1
XS GIS Cut Line= 3
     2341321.463      391042.935     2341351.411      390955.695
     2341523.286      390665.331
#Sta/Elev= 30
       0  732.05    46.1   725.1    65.3  724.01    84.6  721.06    92.2  719.64
   104.2  716.16     120   712.3   135.9  707.35   143.8  704.22   147.8  702.31
   175.6  686.31   179.6  684.43   183.5  683.52   187.5  683.31   199.4  683.92
   202.3  684.91   207.4  687.48   211.3  688.19     247  689.86   270.9  689.34
   286.8  689.51   298.7  690.37   326.4  691.32   338.4  692.56   342.3  693.43
   350.3  696.18     378  707.95   397.9  715.05   413.8  719.58   429.7  722.34
#Mann= 3 ,-1 , 0
       0     .12       0   179.6    .045       0   202.3     .12       0
Bank Sta=179.6,202.3
XS Rating Curve= 0 ,0
Exp/Cntr=0.3,0.1

Type RM Length L Ch R = 1 ,12674.6 ,452,468.5,529.9
XS GIS Cut Line= 3
     2341540.213      391141.893     2341715.994      390786.424
     2341676.932      390709.602
#Sta/Elev= 30
       0  729.18    63.4  713.95    79.3  711.39    91.2   708.6     111  705.64
   126.9  702.45   138.8  699.26   166.6  690.53   174.5   688.6   190.4   687.2
   210.2  687.62   222.1  687.12     230  685.24     234  683.12   237.9  682.08
   253.8  681.88   257.8  681.96   266.1  683.56   273.6  685.74   285.5  686.81
   309.3  685.81   325.2  685.97   333.1  687.37     349  688.32   364.8  690.69
   384.7   692.7   400.5  691.51   416.1  694.56   467.1  697.23   482.7  699.59
#Mann= 3 ,-1 , 0
       0     .12       0     234    .045       0   266.1     .12       0
#XS Ineff= 2 , 0
                          290.12           688.1
Permanent Ineff=
       F       F
Bank Sta=234,266.1
XS Rating Curve= 0 ,0
Exp/Cntr=0.3,0.1

Type RM Length L Ch R = 1 ,12206.1 ,500.4,505.1,508.5
XS GIS Cut Line= 5
      2341713.39      391253.872      2341874.79      391149.929
     2341891.787      391147.432     2342115.734      390994.758
      2342182.14      390994.758
#Sta/Elev= 30
       0  727.11      28  720.87      44  718.65      64  713.92      84  708.38
     108  699.32     116  695.21     132  685.89     136  683.92     140  682.89
     148  682.51     172  683.86     189  679.64   198.8   678.9   213.1  679.48
   225.1   682.6   229.1  683.06     257  682.67   276.9  683.02   284.9  682.58
   296.8  683.57   328.7  682.83   368.6  687.66   376.6  690.29   388.5  695.51
   432.4  719.53   464.2  734.02   484.1  741.31   507.5  748.67   546.6  759.13
#Mann= 3 ,-1 , 0
       0     .12       0     189    .045       0   213.1     .12       0
Bank Sta=189,213.1
XS Rating Curve= 0 ,0
Exp/Cntr=0.3,0.1
